HEC-RAS study SPRINGCK.prj: SPRINGCK

--- SPRINGCK.g01 (geometry) --- (continued)

Type RM Length L Ch R = 1 ,77860   ,589.1,602.3,611.8
XS GIS Cut Line= 2
2151557.59476164386489.4728184792151160.29667172385408.249915317
#Sta/Elev= 30
       0 2333.67    39.2 2322.28    91.6 2298.13   147.5 2267.71   269.4 2214.46
   318.8 2195.14   458.6 2150.24   493.6 2135.87   514.6 2118.37   535.5 2116.81
   550.6 2106.06  562.862101.187     581 2099.34   609.4 2099.81   618.52102.422
   637.5 2114.11   657.9 2117.74   682.3 2131.56   720.8 2134.33   780.2 2149.69
   906.4 2196.89   961.6 2222.24   975.9 2226.39   986.4 2234.86   996.9 2236.83
  1029.1 2257.37  1066.9 2275.96  1101.8 2288.39  1143.7 2306.98  1151.9 2308.35
#Mann= 5 ,-1 , 0
       0      .1       0  514.17     .06       0  562.86    .045       0
   618.5     .06       0  618.68      .1       0
Bank Sta=562.86,618.5
XS Rating Curve= 0 ,0
Exp/Cntr=0.3,0.1

Type RM Length L Ch R = 1 ,77258   ,547,538.7,527
XS GIS Cut Line= 2
2151925.65012789386482.5282785592151971.48369764385375.583970144
#Sta/Elev= 30
       0  2371.5    56.1 2343.07      89 2322.56   131.7 2293.11   164.5 2268.07
   167.8  2265.1   177.6 2252.11   190.8 2241.02   200.9 2230.35   340.7 2142.25
     368 2127.46   391.1 2117.77   420.6 2111.22   459.5 2107.84   513.1 2105.81
   525.7 2102.25   545.4 2101.74  563.782098.114     575 2095.39   604.5 2095.28
  626.062097.973   640.6 2107.06   660.3  2110.6   673.5  2121.7   705.4 2139.96
     726 2149.84   811.4 2178.13   837.6 2188.74   897.8 2209.41  1107.9 2289.74
#Mann= 5 ,-1 , 0
       0      .1       0  520.96     .06       0  563.78    .045       0
  626.06     .06       0  634.34      .1       0
Bank Sta=563.78,626.06
XS Rating Curve= 0 ,0
Exp/Cntr=0.3,0.1

Type RM Length L Ch R = 1 ,76719   ,611.6,597.8,581.6
XS GIS Cut Line= 2
2152653.42819989386474.1949618912152307.59457397385346.417361811
#Sta/Elev= 30
       0 2316.95    46.5 2291.84   130.7 2259.15   149.1 2246.76   170.1 2245.87
   252.4 2217.61   317.1 2201.66   334.8 2200.43   365.7 2204.32   382.8 2201.54
   405.1 2179.97   430.9 2159.11   495.7 2115.04   502.9  2112.5   540.7 2110.59
   547.5 2106.93  560.32 2094.78   568.1 2091.28   595.6 2090.53   619.32093.537
   636.8 2100.38   650.5 2100.14   657.3 2102.55   712.3 2109.06   842.7  2142.2
   904.4 2162.63  1038.3 2217.82    1084 2234.23  1134.3 2249.34  1179.6    2258
#Mann= 4 ,-1 , 0
       0    .055       0  510.08     .06       0  560.32    .045       0
   619.3      .1       0
Bank Sta=560.32,619.3
XS Rating Curve= 0 ,0
Exp/Cntr=0.3,0.1

Type RM Length L Ch R = 1 ,76121   ,498.3,527.6,545.6
XS GIS Cut Line= 2
2153352.03900738385960.306225896 2152456.2058253  385132.5283539
#Sta/Elev= 30
       0 2200.88     106 2169.55   212.3 2131.23   255.2 2119.17   294.5 2099.87
   317.8 2099.25   332.1 2096.51   362.3  2094.5   499.3 2093.93   536.5 2092.23
  550.842088.813     559 2086.58   589.9 2085.52   601.5 2085.68  609.862088.263
   623.2 2092.35   632.9 2097.72   647.9 2100.02   673.4 2118.65   694.3 2130.58
   715.3 2138.77   738.4 2157.15   768.6 2173.71   889.1 2233.45   903.6 2239.32
     961  2251.5  1019.7 2252.39  1077.7 2259.61    1155 2278.53  1219.7 2298.84
#Mann= 7 ,-1 , 0
       0    .055       0  221.83     .06       0  356.38     .06       0
  413.25      .1       0   530.4      .1       0  550.84    .045       0
  609.86      .1       0
Bank Sta=550.84,609.86
XS Rating Curve= 0 ,0
Exp/Cntr=0.3,0.1

Type RM Length L Ch R = 1 ,75594   ,692.1,681.1,657.7
XS GIS Cut Line= 2
 2153396.4834723385961.6950026452153364.53931047384861.694906056
#Sta/Elev= 30
       0 2198.14    43.8 2178.29     151 2145.47   250.6 2107.64   260.4 2105.35
   273.6 2096.77   286.7    2097   312.9  2092.8   355.6 2091.23     402 2086.95
   509.9 2085.88  543.682082.006   555.8 2078.81   578.8 2078.41   595.2 2078.68
  605.912081.571   614.9 2084.12   625.3 2090.71   642.4 2092.55   650.8 2095.83
     658 2101.16   682.7 2113.73   742.9 2151.47   782.3 2168.97   795.4 2171.67
   877.8 2198.05   934.6 2219.16   995.6 2238.66  1038.3 2251.27  1100.5 2266.27
#Mann= 8 ,-1 , 0
       0    .055       0  115.88      .1       0  265.04     .06       0
  388.05     .05       0  543.68    .045       0  605.91      .1       0
  827.49      .1       0  956.66      .1       0
#XS Ineff= 2 , 0
          451.61 2096.48
Permanent Ineff=
       F       F
Bank Sta=543.68,605.91
XS Rating Curve= 0 ,0
Exp/Cntr=0.3,0.1

Type RM Length L Ch R = 1 ,74913   ,460.6,444.1,418.1
XS GIS Cut Line= 2
2154307.50658464385857.2683742342153729.33680922384839.092917144
#Sta/Elev= 30
       0 2370.46    69.9 2371.67     100 2364.92   134.5 2349.67   232.1 2287.56
   243.4 2273.91   257.2 2264.42   271.6 2244.26     315 2213.07   348.6 2179.29
   386.8 2151.45   402.9 2134.91     421 2121.41   434.3 2106.63     464 2102.49
     493  2079.6   518.22075.245   538.7 2073.29  587.082074.946   750.5 2078.76
   781.8 2083.24   793.1 2087.58   816.9 2104.28   832.9 2107.56   847.1 2117.67
   863.6 2123.81   899.7 2133.57   935.8 2136.52   967.8 2143.63  1170.9 2208.78
#Mann= 8 ,-1 , 0
       0      .1       0  377.34     .06       0   518.2    .045       0
  587.08      .1       0  915.71      .1       0     946      .1       0
 1094.28      .1       0 1163.65      .1       0
#XS Ineff= 2 , 0
                          729.12         2083.12
Permanent Ineff=
       F       F
Bank Sta=518.2,587.08
XS Rating Curve= 0 ,0
Exp/Cntr=0.3,0.1

Type RM Length L Ch R = 1 ,74469   ,545.2,555.6,563.7
XS GIS Cut Line= 5
2154733.85481331385370.9386382252154305.95540664385039.677817807
2154287.24415797385032.6158240592154268.53323738385025.551861808
2153779.81702322 384720.02852273
#Sta/Elev= 30
       0 2421.01    26.2 2412.14    44.4 2401.24    59.4 2387.77     109 2351.06
   141.7 2322.64   225.4  2265.9   249.3 2240.96   287.6 2213.02   312.4 2191.39
   408.8 2126.35   464.4 2093.83   504.2 2077.56   528.2 2076.86  541.142070.963
   553.3    2066   575.8 2065.58  607.342069.593   737.1 2073.21   756.1 2078.63
     768 2078.98   776.5 2083.45   796.6  2104.4   811.3 2113.02   884.7 2128.81
   909.2 2139.84   935.1 2141.85   946.7 2147.85  1016.4 2170.52  1157.5 2223.47
#Mann= 4 ,-1 , 0
       0      .1       0  459.15     .06       0  541.14    .045       0
  607.34      .1       0
#XS Ineff= 2 , 0
                          720.71         2076.98
Permanent Ineff=
       F       F
Bank Sta=541.14,607.34
XS Rating Curve= 0 ,0
Exp/Cntr=0.3,0.1

Type RM Length L Ch R = 1 ,73913   ,538.5,537.6,532.6
XS GIS Cut Line= 5
2154862.22594763384902.7784853132154459.11848614384509.764835641
2154445.46168931384495.1533163042154431.86165088384480.489303648
2154025.89034997384103.245635554
#Sta/Elev= 30
       0 2300.54    32.6 2286.45      57 2272.56   102.2 2250.58   115.6 2241.12
   134.6 2224.33   190.3 2187.49   270.6 2126.04   299.4 2108.19   317.9 2094.62
   329.5 2089.97   343.4 2078.42   352.7 2072.63   399.1 2068.75   506.1 2067.77
  546.622062.135   584.5 2060.27   594.6  2060.8  602.992063.906   613.1 2070.02
   628.9 2073.62   655.4 2093.11     738 2118.83   814.6 2146.24   900.5 2181.24
   939.9 2199.56  1007.3 2226.48  1132.5 2284.49  1142.2 2286.64  1157.2 2292.82
#Mann= 5 ,-1 , 0
       0      .1       0  336.26     .06       0   467.9      .1       0
  546.62    .045       0  602.99      .1       0
Bank Sta=546.62,602.99
XS Rating Curve= 0 ,0
Exp/Cntr=0.3,0.1

Type RM Length L Ch R = 1 ,73375   ,576.7,579.3,583.8
XS GIS Cut Line= 2
2155287.09616089 384546.724407392154427.12543988383795.493298307
#Sta/Elev= 30
       0 2224.93    50.2 2214.12   147.9 2200.61   227.9 2187.22   343.9 2161.39
   399.3 2140.12   424.2  2127.8   476.7 2099.35     504 2072.51   525.5 2069.81
  543.132057.174   548.7  2055.2   563.8 2054.89  588.942056.171   605.3 2057.86
   623.2 2063.08   651.1 2063.52     672 2066.94   755.7 2066.45   795.2 2069.49
   814.4 2073.42   910.2 2108.87   949.4 2125.97   962.8  2128.4   971.2 2133.89
  1027.9  2163.5  1048.7 2177.66  1063.9 2190.26  1123.7 2228.63  1141.9 2238.02
#Mann= 5 ,-1 , 0
       0      .1       0  519.58     .06       0  543.13    .045       0
  588.94     .06       0  591.97      .1       0
Bank Sta=543.13,588.94
XS Rating Curve= 0 ,0
Exp/Cntr=0.3,0.1

Type RM Length L Ch R = 1 ,72796   ,538.1,540.6,537.6
XS GIS Cut Line= 2
2155513.24433064383968.9683450612154606.47416255383296.867327064
#Sta/Elev= 30
       0 2293.32    20.7 2290.83    48.5 2282.36    97.5 2256.17   117.9 2242.34
   162.8 2223.15   203.7 2194.13   240.4 2162.23   264.9  2144.2   398.3 2075.29
     416  2068.2   429.5 2065.25   518.1 2060.99  533.272053.953   555.5 2050.42
     600 2050.91  615.062053.995   648.8 2061.13   697.8 2063.11   740.8 2076.15
   795.8 2099.63   808.1  2106.9   816.2 2108.71   836.7    2119   853.3  2129.7
   865.1 2132.94   987.8  2194.8  1001.1 2198.52  1062.1 2228.62  1128.7 2257.34
#Mann= 4 ,-1 , 0
       0      .1       0  463.04    .055       0  533.27    .045       0
  615.06      .1       0
Bank Sta=533.27,615.06
XS Rating Curve= 0 ,0
Exp/Cntr=0.3,0.1

Type RM Length L Ch R = 1 ,72256   ,557.3,555.2,555.1
XS GIS Cut Line= 2
2155685.23644072383477.0693944842154784.40556522 382763.94418031
#Sta/Elev= 30
       0 2354.05    26.6 2338.63   160.2 2240.37   194.6 2220.15   214.6 2201.83
   260.7 2173.24   319.3 2132.95   377.8 2085.33   400.1 2071.17   415.5 2063.97
   432.2 2059.84   515.9 2057.32  533.552049.848   555.2 2046.07   595.4  2046.3
  605.562049.225     622 2054.99   641.5  2057.7   670.7 2074.95   779.5 2128.13
   792.1 2130.17   827.5 2148.13     909 2183.57   919.9 2184.96   934.4  2192.8
   986.4 2208.97  1033.1  2231.3  1046.8 2234.09    1089 2256.21  1148.9 2280.37
#Mann= 5 ,-1 , 0
       0      .1       0  489.33     .06       0  530.03      .1       0
  533.55    .045       0  605.56      .1       0
Bank Sta=533.55,605.56
XS Rating Curve= 0 ,0
Exp/Cntr=0.3,0.1

Type RM Length L Ch R = 1 ,71700   ,612,607.3,601.7
XS GIS Cut Line= 2
2155908.06539139382946.8322659732154985.21848381382263.517359644
#Sta/Elev= 30
       0  2342.1    33.5 2319.77   164.2 2248.26   261.8 2189.08   362.7 2117.37
   392.8 2094.41   411.9 2076.18   432.3 2061.93   458.1 2053.12   515.2  2051.6
  528.21 2046.63   543.8 2043.24   576.1 2042.87   592.6 2043.95  600.392046.677
   621.4 2054.03   678.5 2054.33   691.1 2058.71   723.4 2075.78   761.4 2090.29
   809.2  2099.8   859.9 2119.49   897.5 2128.43   943.9 2147.85   984.7 2169.19
  1054.1 2199.15  1070.4 2210.36  1082.8 2210.62  1106.2 2225.29  1148.3 2237.74
#Mann= 4 ,-1 , 0
       0      .1       0  460.96     .06       0  528.21    .045       0
  600.39      .1       0
#XS Ineff= 2 , 0
                          624.79         2060.24
Permanent Ineff=
       F       F
Bank Sta=528.21,600.39
XS Rating Curve= 0 ,0
Exp/Cntr=0.3,0.1

Type RM Length L Ch R = 1 ,71093   ,589.7,586.4,580.5
XS GIS Cut Line= 2
2156166.07274939382331.1829067322155178.76665314381755.800855398
#Sta/Elev= 30
       0 2359.11    20.7 2348.15    37.4 2335.83    71.1  2323.6   104.6 2300.02
   284.3 2197.93   356.4 2151.89   398.2 2128.37   458.9 2078.71   487.1 2061.02
   500.7 2048.26   522.1 2046.49  533.712042.353   542.5 2039.45   567.7 2038.83
  589.372040.507   603.2 2040.68   622.2    2048   637.3 2048.67   652.6 2056.87
   706.8 2069.44   780.4 2076.24   843.6 2089.69     907 2118.65   969.3 2131.16
  1058.9 2158.83  1086.6 2169.85  1112.3 2184.62  1127.3 2188.32  1142.7 2197.91
#Mann= 5 ,-1 , 0
       0      .1       0  471.35     .06       0  533.71    .045       0
  589.37     .06       0  603.72      .1       0
Bank Sta=533.71,589.37
XS Rating Curve= 0 ,0
Exp/Cntr=0.3,0.1

Type RM Length L Ch R = 1 ,70507   ,569.2,571.2,570.2
XS GIS Cut Line= 3
2156394.08902563381732.3379758152156046.86662297381562.893432811
2155306.38647664381291.956638724
#Sta/Elev= 30
       0 2264.72    92.6 2230.41   194.8 2211.92     237 2200.49   251.7 2191.79
   278.7 2187.69   305.7 2175.95   338.4 2151.47   369.5 2143.68   423.1 2120.38
   454.6 2113.66   468.6 2103.78   510.5 2084.66   531.4 2062.27   555.9 2060.03
   573.3 2043.63  582.672038.758   594.3 2035.36   611.9  2035.1   632.7 2035.16
  644.83 2038.59   665.4 2044.02   737.5 2046.96   758.5 2044.06   839.4 2062.04
   898.2  2083.8   946.8 2105.12  1097.4  2159.9  1136.1 2177.52  1174.9  2198.9
#Mann= 4 ,-1 , 0
       0      .1       0  483.89     .06       0  582.67    .045       0
  644.83      .1       0
#XS Ineff= 2 , 0
                          736.16         2054.65
Permanent Ineff=
       F       F
Bank Sta=582.67,644.83
XS Rating Curve= 0 ,0
Exp/Cntr=0.3,0.1

Type RM Length L Ch R = 1 ,69935   ,551.8,557,562.5
XS GIS Cut Line= 2
2156288.53346246381217.060134977 2155232.9778308 380754.56007573
#Sta/Elev= 30
       0 2143.92    68.7 2118.18   147.8 2083.34   197.7 2063.94   254.9 2048.51
   276.5  2048.6   385.7 2042.45   473.5 2042.39   530.8 2040.27   541.5 2041.34
   566.3 2039.33  589.31 2034.24   609.6 2030.08   634.7 2030.26  648.242034.985
   658.4 2041.98   670.5 2043.72     717 2081.36   777.9 2123.58   843.5 2158.86
   874.6 2183.13   896.1 2196.92   933.4 2224.64   989.7 2260.66  1025.1 2288.84
    1032 2292.23    1043 2294.78  1064.4 2308.41  1111.1 2331.11  1152.4 2353.85
#Mann= 5 ,-1 , 0
       0      .1       0  212.73     .06       0  406.14      .1       0
  589.31    .045       0  648.24      .1       0
#XS Ineff= 2 , 0
          549.22 2053.92
Permanent Ineff=
       F       F
Bank Sta=589.31,648.24
XS Rating Curve= 0 ,0
Exp/Cntr=0.3,0.1

Type RM Length L Ch R = 1 ,69378   ,599.3,604.3,607.9
XS GIS Cut Line= 2
2156419.12506481380810.4946751452155488.53342205380124.004578307
#Sta/Elev= 30
       0 2135.72    52.2 2119.87     132 2099.28     207 2076.67   228.3 2069.24
   244.6 2060.93   249.3 2058.09   263.3 2046.58   285.3 2045.42   301.6 2038.01
   407.6    2036     512 2037.31   523.8 2033.65   548.6 2028.32  570.012027.722
     587 2026.53   607.4 2026.83  619.152029.514   624.7 2032.11   635.9 2040.37
   650.5 2044.04   666.9 2060.16   741.9 2100.37   775.1 2115.23     864 2149.52
   924.4  2178.8   953.1 2191.22   974.3 2201.67  1030.5 2233.23  1156.4 2296.25
#Mann= 6 ,-1 , 0
       0      .1       0   209.2     .06       0   333.4     .05       0
  505.94      .1       0  570.01    .045       0  619.15      .1       0
#XS Ineff= 2 , 0
          504.77 2036.82
Permanent Ineff=
       F       F
Bank Sta=570.01,619.15
XS Rating Curve= 0 ,0
Exp/Cntr=0.3,0.1

Type RM Length L Ch R = 1 ,68774   ,564.3,566,565.6
XS GIS Cut Line= 2
2156720.00963363380396.8170248122155966.42682321 379643.21748215
#Sta/Elev= 30
       0 2122.04    61.1 2105.76   179.5 2079.76   244.5 2060.19   254.9 2053.39
   275.8  2052.9   288.4 2048.41   311.6 2043.46   398.7 2031.92   442.8 2030.73
   514.7 2033.01   529.7 2031.73   548.3 2025.73  560.742025.049   588.9 2022.73
   608.6    2023  619.772027.112   645.7 2039.94   653.9 2048.36   667.8 2071.78
     676 2080.32   696.7 2096.03   716.5 2108.96   759.5 2132.06   881.2 2187.61
   905.5 2196.07   927.6 2201.65     973 2203.16  1028.6  2202.5  1065.7  2205.2
#Mann= 6 ,-1 , 0
       0      .1       0  201.58     .06       0   322.4     .05       0
  510.34      .1       0  560.74    .045       0  619.77      .1       0
#XS Ineff= 2 , 0
          517.49 2034.23
Permanent Ineff=
       F       F
Bank Sta=560.74,619.77
XS Rating Curve= 0 ,0
Exp/Cntr=0.3,0.1

Type RM Length L Ch R = 1 ,68208   ,557.5,555.5,546.9
XS GIS Cut Line= 3
2157169.20460139380120.2342446452156878.92696673379771.623393312
2156336.86604297379193.811884895
#Sta/Elev= 30
       0 2103.66      39 2095.09    64.7 2092.63   126.2 2083.79   144.6 2078.62
   195.8 2075.81   208.6 2072.06   238.5 2067.63   285.3 2056.97   310.9 2053.15
   385.5 2048.58   488.1 2032.29   514.9 2030.51     579 2029.15   603.9 2023.48
  620.612022.745   640.8 2021.85   675.9 2022.04  686.082024.444   703.8 2027.12
   712.8 2030.09   729.3 2030.81     778 2054.91   945.1 2117.53  1014.7 2146.85
  1121.5  2188.9  1149.6 2198.01  1177.2 2205.14    1212 2210.09  1245.9 2211.47
#Mann= 6 ,-1 , 0
       0     .05       0   81.16     .06       0  273.94     .05       0
  500.42      .1       0  620.61    .045       0  686.08      .1       0
Bank Sta=620.61,686.08
XS Rating Curve= 0 ,0
Exp/Cntr=0.3,0.1

Type RM Length L Ch R = 1 ,67653   ,481.6,472.7,465.1
XS GIS Cut Line= 2
2157700.51095347379655.2108964772156678.92703864  378971.6233529
#Sta/Elev= 30
       0 2178.94    57.5 2161.69   138.8 2134.28     160 2121.95   183.6  2120.1
   195.5 2111.97   231.1 2092.41   271.2 2072.78   349.3 2048.47   401.3 2026.81
   452.2 2024.83   566.8 2027.31   578.9 2026.22  586.74 2020.82   590.5 2017.54
   597.6 2016.42  639.182020.537   661.4 2023.69   673.3 2022.28   689.1 2025.23
   722.9 2023.46   787.8 2027.05   862.5 2025.66   874.3 2032.16   885.7 2035.09
   910.1 2047.64   961.4 2069.13    1073  2109.6  1168.8 2148.19  1229.2 2167.41
#Mann= 7 ,-1 , 0
       0     .05       0  102.15     .06       0  284.27      .1       0
  356.27     .05       0   495.8      .1       0  586.74    .045       0
  639.18      .1       0
#XS Ineff= 2 , 0
                          764.57          2034.6
Permanent Ineff=
       F       F
Bank Sta=586.74,639.18
XS Rating Curve= 0 ,0
Exp/Cntr=0.3,0.1

Type RM Length L Ch R = 1 ,67180   ,725.2,723.1,718.1
XS GIS Cut Line= 2
2158049.13624047379111.2766169012156860.12877597378750.660868317
#Sta/Elev= 30
       0 2177.17    13.1 2175.56    23.4 2166.16    30.2  2162.3   122.8 2124.67
     174 2101.27   239.4 2064.04   273.6 2036.87   287.1 2029.38   301.1 2023.93
   318.2 2020.41   338.8 2019.18   558.2 2021.56  580.272018.013   589.1 2015.97
   619.9 2015.23     6362017.333   643.9 2017.08   681.6 2022.69   777.6 2020.68
   835.9 2021.33   860.6 2023.74   880.5 2030.55   935.3 2059.48   953.3 2067.39
   968.4 2071.84  1000.5 2077.98  1073.7 2087.45  1144.5 2098.78  1242.5 2116.68
#Mann= 8 ,-1 , 0
       0     .06       0   27.13      .1       0  197.58      .1       0
  252.76     .05       0  507.43      .1       0  580.27    .045       0
     636      .1       0 1185.33     .05       0
#XS Ineff= 1 ,-1
  774.87 1242.49 2027.14
Permanent Ineff=
       F
Bank Sta=580.27,636
XS Rating Curve= 0 ,0
Exp/Cntr=0.3,0.1

Type RM Length L Ch R = 1 ,66457   ,560.9,561.8,565.5
XS GIS Cut Line= 5
2158219.06897147378378.2679123132157648.52352464378239.022455901
2157628.78471898378235.8003494742157609.04591331378232.578243062
 2157029.3758128378139.242799804
#Sta/Elev= 30
       0 2167.37    39.2 2155.74    49.3 2146.62    52.7 2145.23    76.4 2142.48
    89.9 2134.88   170.9 2102.83   204.7 2087.42   238.5 2070.38   268.9 2052.17
   295.9 2032.94   309.4 2018.45   316.1  2015.6   339.8 2014.43   549.2 2017.48
   569.4 2016.16  580.772012.412   589.6 2010.16   622.1 2009.81  640.412013.225
   649.5 2016.35     665 2017.82     686 2026.03   795.7 2026.67     830 2028.42
   938.6 2038.99  1065.7 2042.54  1102.9 2045.22  1144.6  2051.2  1214.4 2068.44
#Mann= 8 ,-1 , 0
       0     .06       0  124.69      .1       0  232.54      .1       0
   364.7     .05       0  561.15      .1       0  580.77    .045       0
  640.41      .1       0   743.4     .05       0
Bank Sta=580.77,640.41
XS Rating Curve= 0 ,0
Exp/Cntr=0.3,0.1

Type RM Length L Ch R = 1 ,65895   ,599,590.5,573.4
XS GIS Cut Line= 2
2158381.53190114377859.9352875652157115.84250338377515.755201638
#Sta/Elev= 30
       0 2140.88      65 2123.72   214.6 2079.76   224.7 2075.89   238.4 2067.76
   248.6 2064.39   276.5 2062.69   357.4 2053.75   377.8 2050.03   401.6 2043.27
   418.6 2033.59     439 2030.72   449.2 2024.49   462.8 2012.89   544.4 2013.18
  557.452011.913   568.2 2008.86   584.7 2008.41   615.8 2008.48  629.592010.658
   646.4 2013.53   666.8 2012.77   700.5 2015.79   840.2 2014.17   979.6 2016.03
    1068 2015.52  1159.8 2018.29  1214.2 2024.87  1251.6 2032.51  1311.7 2053.83
#Mann= 5 ,-1 , 0
       0      .1       0  557.45    .045       0  629.59      .1       0
  651.54     .05       0 1277.22      .1       0
#XS Ineff= 2 , 0
                          958.41        2023.919
Permanent Ineff=
       F       F
Bank Sta=557.45,629.59
XS Rating Curve= 0 ,0
Exp/Cntr=0.3,0.1

Type RM Length L Ch R = 1 ,65304   ,548.2,539,526
XS GIS Cut Line= 2
2158483.77546306 377111.825891392157111.67584506377165.755245477
#Sta/Elev= 30
       0 2153.95    79.8 2118.47   171.5 2071.72   230.8 2045.66   270.2 2042.85
   309.6  2045.4     333 2044.06   365.4 2037.62   431.1 2016.51   477.1 2014.15
   506.6    2011   516.5 2008.01     527 2003.89     569 2003.61   601.8 2008.27
   621.5 2013.23   667.5 2010.88   937.1 2010.22   976.1 2010.89  1012.2 2015.75
  1038.5 2016.94    1091 2017.09  1160.7 2014.02  1224.2 2015.75  1249.1 2019.17
  1268.1 2024.62  1307.7 2040.93  1327.4 2044.03  1353.7 2060.36  1373.2 2069.76
#Mann= 6 ,-1 , 0
       0      .1       0  450.22      .1       0   516.5    .045       0
   601.8      .1       0  658.78     .05       0 1222.46      .1       0
Bank Sta=516.5,601.8
XS Rating Curve= 0 ,0
Exp/Cntr=0.3,0.1

Type RM Length L Ch R = 1 ,64765   ,683.1,660.7,630.9
XS GIS Cut Line= 2
2158299.17576663376451.1720289742157226.25894922376803.255314305
#Sta/Elev= 30
       0 2303.76    24.3 2287.38    45.5 2268.92    76.1 2244.69   100.2 2221.76
   110.6 2214.35   138.2 2186.75   155.5  2172.6   217.6 2125.96   255.6 2099.57
   299.5 2072.18     373 2030.95     411 2018.17   428.3 2009.47  468.052003.872
   476.6 2002.18   493.9 2002.11   524.9 2002.33  540.062005.496   580.2 2009.02
   645.8 2007.15     777  2006.6   915.1 2007.58   942.8 2008.93   949.7 2009.82
   973.8 2027.09  1001.5 2038.56    1049    2044  1078.2 2051.15  1129.2 2055.58
#Mann= 5 ,-1 , 0
       0      .1       0  468.05    .045       0  540.06      .1       0
  547.61     .05       0  929.01      .1       0
Bank Sta=468.05,540.06
XS Rating Curve= 0 ,0
Exp/Cntr=0.3,0.1

Type RM Length L Ch R = 1 ,64105   ,573.1,570.8,565.8
XS GIS Cut Line= 2
2157498.30761772375902.1396624742157164.97429489376760.473247647
#Sta/Elev= 30
       0 2254.88    27.2 2223.65    45.1 2206.92    62.7 2193.31    72.8 2177.48
    80.3 2168.23   114.5 2138.76   161.6 2091.62   168.3 2081.45   178.8    2060
   182.4 2054.42   202.1 2032.12   217.6 2017.51  229.382001.453   235.2 1999.09
   260.4 1998.55  278.532002.351     295 2004.22   326.7 1998.23   340.7 1997.69
   358.3 1998.78   375.9 2006.33   492.1 2003.29     566 2005.94   651.8  2003.7
   805.3 2007.63   840.5  2013.5   860.3 2022.95   886.3  2038.9   920.8 2048.25
#Mann= 5 ,-1 , 0
       0      .1       0  229.38    .045       0  278.53      .1       0
  481.13     .05       0  744.49      .1       0
Bank Sta=229.38,278.53
XS Rating Curve= 0 ,0
Exp/Cntr=0.3,0.1

Type RM Length L Ch R = 1 ,63534   ,665.3,674.5,689.8
XS GIS Cut Line= 2
2156909.70807314 375765.855158152156720.17105064376710.299463481
#Sta/Elev= 30
       0 2086.51      92 2053.91   121.6 2036.99   145.1 2026.48   175.1 2007.31
   185.2 2002.35   198.6 2000.54   218.7 2001.22   242.1 2000.41   275.6 2002.03
   292.3 2000.25  301.431995.822   305.7 1993.95   322.4 1992.23   342.5 1992.51
   352.5 1994.49  366.961995.924   399.4 2001.39   462.3 1999.52   536.6 1999.33
   677.1 2001.34   710.6 2003.63     724 2008.89     744 2019.27   757.4 2025.01
     824  2051.6   884.6 2074.56     898 2078.83   921.4 2083.76   963.3 2090.12
#Mann= 6 ,-1 , 0
       0      .1       0  298.74      .1       0  301.43    .045       0
  366.96      .1       0  450.07     .05       0  686.17      .1       0
Bank Sta=301.43,366.96
XS Rating Curve= 0 ,0
Exp/Cntr=0.3,0.1

Type RM Length L Ch R = 1 ,62859   ,565.2,552,536.1
XS GIS Cut Line= 3
2156392.39349097375588.771850899 2156192.3932348375897.104895636
2155840.30994947376565.855198562
#Sta/Elev= 30
       0 2105.36   104.8 2051.06   125.6 2041.45   138.2  2036.9   149.8  2029.1
   165.5 2027.33   181.2 2021.64   204.4 2015.11   212.5  2010.9     232 1996.83
  240.681993.556   251.8 1990.66   267.2 1990.31  308.981995.272     323 1997.76
   542.7 1996.12   591.3 1998.03   643.2 1998.02   691.4 1996.09   754.4 1997.66
   817.4 1995.66   921.3 1997.05   928.7 1999.37   947.2 2014.88   973.2 2029.08
    1036  2057.5    1070 2068.59  1084.6  2072.3  1110.4 2076.88  1123.3 2076.76
#Mann= 6 ,-1 , 0
       0      .1       0  240.68    .045       0  308.98      .1       0
  317.73      .1       0  370.18     .05       0 1028.22      .1       0
#XS Ineff= 1 ,-1
  740.92 1123.29 2009.02
Permanent Ineff=
       F
Bank Sta=240.68,308.98
XS Rating Curve= 0 ,0
Exp/Cntr=0.3,0.1

Type RM Length L Ch R = 1 ,62307   ,1104.2,1109.4,1102.4
XS GIS Cut Line= 3
2155771.56008697375345.021682233 2155750.7267953375642.938409224
2155715.30987139 376536.68826215
#Sta/Elev= 30
       0 2095.54    11.9 2094.03   100.7 2059.23   120.4  2048.5   130.3 2044.63
   148.6 2034.29   182.9 2007.01  198.011991.997     206 1988.49   225.7 1988.22
   245.4 1989.63   253.21991.583   261.9 1994.76   281.6 1996.25   350.6 1992.25
   392.9  1994.2     460 1993.68   488.6 1992.09   557.4 1995.78   623.1 1994.41
   700.6 1995.61   764.3 1992.76   882.5 1995.43   938.3 1994.05  1020.4 1997.93
  1030.2 1999.06  1046.7 2005.27    1155 2053.21  1184.6 2065.38  1193.1 2066.59
#Mann= 4 ,-1 , 0
       0      .1       0  198.01    .045       0   253.2      .1       0
  294.13     .05       0
#XS Ineff= 1 ,-1
  755.18 1193.09 2011.06
Permanent Ineff=
       F
Bank Sta=198.01,253.2
XS Rating Curve= 0 ,0
Exp/Cntr=0.5,0.3

Type RM Length L Ch R = 1 ,61198   ,31.4,31.9,32.1
XS GIS Cut Line= 3
2154787.54860355375591.0546547322154743.06083164376099.952258974
2154676.87165955376770.525064811
#Sta/Elev= 30
       0 2188.18    25.1 2174.48      35 2163.29    58.1 2142.19    74.5 2130.11
    87.7 2118.27   153.6 2072.92   193.1 2040.43   212.9 2026.75   268.8 1992.39
   278.7 1989.86   295.7 1988.67   374.2 1989.42  389.681985.346   397.3 1982.11
   409.8 1981.57   430.2 1981.71   438.81985.138   449.2 1989.83   535.6 1986.98
   641.8 1987.76   769.7 1986.09   944.4  1987.9   977.4 1993.92  1026.8 2018.08
  1043.3  2020.6  1056.5 2026.63  1096.1 2039.29  1145.5 2049.64  1184.7 2054.06
#Mann= 4 ,-1 , 0
       0      .1       0  389.68    .045       0   438.8     .06       0
   535.6     .05       0
#XS Ineff= 2 , 0
          379.68  1988.2   448.8          1988.2
Permanent Ineff=
       F       F
Bank Sta=389.68,438.8
XS Rating Curve= 0 ,0
Exp/Cntr=0.5,0.3

Type RM Length L Ch R = 1 ,61166   ,772.7,775.2,776.7
XS GIS Cut Line= 2
2154759.83540438375581.3063146472154647.33562939 376775.05622372
#Sta/Elev= 30
       0 2185.13    18.5 2177.48    28.4 2171.64      58 2144.77   113.9 2103.58
   153.6 2079.31   196.4 2044.73   232.7 2018.95   275.5  1991.9     292 1988.09
   377.7 1988.59  393.131986.202     404 1982.82   439.2 1981.68   446.9 1982.76
   452.11986.515   459.8 1988.44   624.8 1986.12   703.9 1987.19   825.8 1986.03
   941.2  1986.5   977.4 1988.56  1003.8 1995.72  1023.4 2007.51    1040 2015.18
  1056.6 2017.12    1073 2024.65  1099.3 2033.05  1136.5 2040.68    1199 2045.18
#Mann= 6 ,-1 , 0
       0      .1       0  393.13    .045       0   452.1     .06       0
  568.71     .05       0 1022.04      .1       0 1113.57     .05       0
Bank Sta=393.13,452.1
XS Rating Curve= 0 ,0
Exp/Cntr=0.5,0.3

Type RM Length L Ch R = 1 ,60391   ,489.8,528.4,551.6
XS GIS Cut Line= 3
 2154073.7242438 375607.000817062153988.30774798375929.917494059
2153838.30771989376934.084120899
#Sta/Elev= 30
       0 2089.32    73.9 2084.77   196.1 2081.18   219.5 2077.51   260.5 2064.17
   311.4 2051.24   321.6 2047.13   328.4  2046.5   351.8 2037.46   378.3 2024.46
   394.9 2014.06   408.2 2003.01   421.4 1984.87  432.28 1981.56   444.6 1978.84
   461.2 1977.92   481.1 1978.45  491.23 1982.49     511 1984.59   617.1 1983.45
   650.3 1981.66   819.5 1983.48   879.2 1986.39   959.1 1986.29  1018.5 1989.17
  1197.7 1992.91  1237.5 1998.64  1264.6 2004.88  1302.1 2014.48  1349.3 2029.08
#Mann= 5 ,-1 , 0
       0      .1       0  377.57      .1       0  432.28    .045       0
  491.23      .1       0  495.97     .05       0
Bank Sta=432.28,491.23
XS Rating Curve= 0 ,0
Exp/Cntr=0.3,0.1

Type RM Length L Ch R = 1 ,59863   ,570.9,598.9,621
XS GIS Cut Line= 2
2154034.73941363375591.6383149772152971.64114614376113.250788808
#Sta/Elev= 30
       0 2082.48    70.3 2071.34   116.9 2062.39   194.5 2053.82   260.3 2044.77
   344.3 2027.44     359 2025.36   410.1 2011.55   428.4 2003.17     454 1985.69
   461.3 1983.05   545.3  1982.2  551.081980.714     560 1977.05   581.9 1975.16
   600.2 1975.93  616.691980.467     633 1982.19   848.7 1979.72   886.7 1980.39
   901.4  1982.4   925.4 1992.64   998.5 2034.29  1031.4 2054.29  1075.5 2087.81
  1111.8 2118.47  1122.7 2126.29  1131.8 2134.46  1146.6 2144.66  1184.2 2176.08
#Mann= 6 ,-1 , 0
       0      .1       0  459.94      .1       0  551.08    .045       0
  616.69      .1       0  629.83     .05       0  832.89      .1       0
Bank Sta=551.08,616.69
XS Rating Curve= 0 ,0
Exp/Cntr=0.3,0.1

Type RM Length L Ch R = 1 ,59264   ,615.7,612.1,608.3
XS GIS Cut Line= 2
2154063.03463264375562.8319421412152713.75747555375180.496092647
#Sta/Elev= 30
       0 2085.68    30.2 2080.81   129.2 2059.21   231.4 2042.23   282.5 2030.58
     324 2018.44   391.6 1994.96   401.9 1993.44   418.9 1983.25   429.1  1980.5
   701.9 1978.36   733.2 1979.74  747.071976.021   759.9 1972.27   780.8 1971.76
   804.1  1973.1  815.881977.001   841.8 1993.62   889.1 2039.63     927 2068.91
   947.5 2089.74   957.7 2103.08   964.5  2109.5   988.4 2125.14  1032.6 2130.98
  1117.6 2128.23  1189.6 2133.32  1254.4 2150.54  1330.2 2175.44  1402.4 2193.64
#Mann= 5 ,-1 , 0
       0      .1       0   418.4     .05       0  660.12      .1       0
  747.07    .045       0  815.88      .1       0
Bank Sta=747.07,815.88
XS Rating Curve= 0 ,0
Exp/Cntr=0.3,0.1

Type RM Length L Ch R = 1 ,58652   ,632.7,618.4,606.6
XS GIS Cut Line= 2
2154250.53458571374877.0678937292152876.64724164374682.768741637
#Sta/Elev= 30
       0 2080.59      53 2082.67    76.2 2081.59    96.1  2079.4   139.2 2069.86
   255.1 2033.32   292.5 2015.54   308.1 2005.52   347.9 1984.22   370.8 1978.25
   596.4 1976.61   639.5 1974.51   709.1 1976.56   715.7 1975.78  721.66 1973.04
     729 1969.99   735.6 1969.33   768.5 1969.47  780.711973.352   795.2 1986.43
   808.5 1995.85   867.2 2026.84  1007.3 2087.44  1033.8 2095.42  1050.4 2097.33
  1079.1 2097.62  1137.2 2092.67  1166.3 2092.07    1262 2097.96  1387.6 2098.34
#Mann= 5 ,-1 , 0
       0      .1       0  375.68     .05       0  670.52      .1       0
  721.66    .045       0  780.71      .1       0
Bank Sta=721.66,780.71
XS Rating Curve= 0 ,0
Exp/Cntr=0.3,0.1

Type RM Length L Ch R = 1 ,58033   ,1098.6,1114.1,1021.9
XS GIS Cut Line= 2
2154118.58996773373984.7068175672152898.10389164 374321.51257439
#Sta/Elev= 30
       0 2089.88    12.9 2084.83    36.7 2073.38    84.3 2046.44   118.4 2028.25
   196.7 1977.34   206.9 1973.65   217.1 1972.84   332.8  1973.9   390.7 1971.82
   455.3 1973.78   509.8 1973.16   533.6 1972.09   625.5 1974.51  642.891973.035
   652.7 1969.93   700.4 1969.06   707.2 1970.26  711.77 1973.77   720.8  1983.8
   737.8 1994.72   754.6 2003.95   792.2 2020.63   822.9 2030.69   979.5 2066.91
   996.5 2069.09  1102.5 2077.46  1200.4  2089.5  1234.7 2091.78  1266.1 2092.34
#Mann= 5 ,-1 , 0
       0      .1       0  200.93     .05       0  605.06      .1       0
  642.89    .045       0  711.77      .1       0
Bank Sta=642.89,711.77
XS Rating Curve= 0 ,0
Exp/Cntr=0.3,0.1

Type RM Length L Ch R = 1 ,56919   ,772.7,819.6,820.8
XS GIS Cut Line= 3
2153526.57605989373166.9984792322153151.57615373373382.276263893
2152462.33999939373732.970772475
#Sta/Elev= 30
       0  2047.4    35.6 2047.87    73.1 2046.35   126.1 2039.35   165.4 2028.55
   258.5 1994.97   266.1  1990.8     285 1973.84  298.091968.974   315.3 1963.19
   334.2 1963.66   352.9 1961.45   364.4 1964.16   372.1 1964.23  386.541968.981
   405.2 1969.93   619.6 1968.69   676.1 1969.05   688.3 1970.61   704.9 1968.91
   822.5 1968.47   848.5 1969.46   863.2 1973.94   896.4 1979.75   937.2 1979.91
   951.6 1983.06   974.1 1991.16  1066.5 2031.91  1129.9  2054.7  1205.7 2078.41
#Mann= 3 ,-1 , 0
       0      .1       0  298.09    .045       0  386.54      .1       0
Bank Sta=298.09,386.54
XS Rating Curve= 0 ,0
Exp/Cntr=0.3,0.1

Type RM Length L Ch R = 1 ,56100   ,767.3,682.4,626.9
XS GIS Cut Line= 6
2153378.39230114373094.0750686382153036.72566164372784.352590978
2152977.00334014372751.0193243182152824.76939264372709.940010145
2152804.80420947372728.1693044012152547.85984147372996.398426726
#Sta/Elev= 30
       0 2032.44   124.2 2005.14   149.7 1998.16   162.6 1996.26   186.9 1988.02
     200 1980.49   210.1 1979.01   221.2 1974.01   235.4 1971.46   261.2 1969.33
   394.9 1968.23   421.4 1969.59   449.3 1968.53   532.4 1970.42   538.7 1969.61
   552.7 1964.82   593.5 1963.43  600.341961.573   610.5 1958.72   637.7 1958.61
   647.9 1957.25   658.1 1959.26   664.71963.599   675.1 1969.68   699.4 1972.78
   710.6 1979.05   719.9    1982   772.8  1993.3   866.4 2005.85  1085.7    2044
#Mann= 3 ,-1 , 0
       0      .1       0  600.34    .045       0   664.7      .1       0
Bank Sta=600.34,664.7
XS Rating Curve= 0 ,0
Exp/Cntr=0.3,0.1

Type RM Length L Ch R = 1 ,55417   ,575.1,578.8,582.8
XS GIS Cut Line= 3
2152453.67564663372113.9333281372152683.49342847372753.541957065
2152559.36145888 372967.95163323
#Sta/Elev= 30
       0 2215.92    15.6 2209.08      40 2195.32    43.4 2191.32    51.7 2177.74
    60.9 2162.11    64.4 2154.04    67.8 2148.44    77.3 2137.27   113.2 2109.31
   120.9 2101.63   175.9  2054.9   207.3    2032   280.5 1967.32  287.541962.098
     291 1959.25   297.9 1957.06   332.8 1955.98   350.2 1956.82  362.691960.497
   385.1    1961   402.5 1964.81   437.4 1963.04   538.5 1963.91   632.6 1968.14
   667.5 1974.41   681.7 1980.74     746  1991.6   818.6    2006   927.4 2034.29
#Mann= 3 ,-1 , 0
       0      .1       0  287.54    .045       0  362.69      .1       0
Bank Sta=287.54,362.69
XS Rating Curve= 0 ,0
Exp/Cntr=0.3,0.1

Type RM Length L Ch R = 1 ,54838   ,491.3,496.6,500.6
XS GIS Cut Line= 2
2151929.76068397372209.791732222 2152150.5942318 373182.01419723
#Sta/Elev= 30
       0 2077.56    24.4 2068.65    31.1 2064.54    41.2 2063.43    51.3 2059.95
    84.9 2044.45   105.9 2037.89   145.5 2029.79   280.1 1987.26   312.9 1971.93
   337.3 1957.79     344 1956.95   378.2 1959.71  400.111957.447   411.3  1954.1
   428.1  1953.6   451.6 1954.04   465.71958.299   498.7 1959.23   522.3 1962.27
   539.1 1961.03   582.9 1962.85   757.8  1961.5   801.5  1963.8   825.1 1978.77
   841.9 1991.41     918 2039.06     963  2071.7   979.9 2078.22     997 2088.41
#Mann= 3 ,-1 , 0
       0      .1       0  400.11    .045       0   465.7      .1       0
Bank Sta=400.11,465.7
XS Rating Curve= 0 ,0
Exp/Cntr=0.3,0.1

Type RM Length L Ch R = 1 ,54342   ,745.5,763,775.2
XS GIS Cut Line= 2
 2151596.1012463372296.1390004752151512.76775156373306.555614814
#Sta/Elev= 30
       0  2098.5      59 2086.94   105.1 2072.58   111.7 2069.26   124.8 2067.54
   236.8 2015.38   292.7 1985.52   315.8  1970.9   332.2 1957.86   348.7    1953
     366 1956.19   394.8 1957.53  451.331954.657   483.7 1953.34     487 1953.58
  490.571956.647   500.1 1958.37   526.5 1955.99   539.6 1959.33   562.7 1959.77
   707.5 1959.12   733.9 1962.74   778.6 1995.59   835.3  2039.9     859 2060.66
   921.5 2099.84   954.4 2126.56   980.8 2139.45   990.6 2150.07  1013.8 2165.78
#Mann= 3 ,-1 , 0
       0      .1       0  451.33    .045       0  490.57      .1       0
Bank Sta=451.33,490.57
XS Rating Curve= 0 ,0
Exp/Cntr=0.3,0.1

Type RM Length L Ch R = 1 ,53579   ,673.1,698,715.7
XS GIS Cut Line= 3
2151073.18431313372221.1391504712150804.43452255372577.389094144
2150537.76773305373054.472457558
#Sta/Elev= 30
       0 2047.46      57 2039.59     139    2020     153 2013.06   164.7 2011.52
   175.8 2005.08     221 1989.19   245.7 1976.88   274.8  1957.9     332 1955.79
  338.761952.919   344.3 1950.21     392 1948.79  403.911952.989   410.1 1955.55
   443.5 1956.36   589.8 1953.72   625.3 1958.36   653.2 1976.93   698.8 2015.67
   739.6 2046.26   759.8 2058.68     789 2084.67   802.6 2092.94   815.3 2105.11
   831.6 2115.12   868.7 2143.71   946.9 2191.36   961.9 2203.12   992.8 2212.98
#Mann= 3 ,-1 , 0
       0      .1       0  338.76    .045       0  403.91      .1       0
Bank Sta=338.76,403.91
XS Rating Curve= 0 ,0
Exp/Cntr=0.3,0.1

Type RM Length L Ch R = 1 ,52881   ,591,601.7,589
XS GIS Cut Line= 3
2151071.10098398371891.9724859742150748.18430696371910.722448483
2150022.11358064372072.812019303
#Sta/Elev= 30
       0 2042.58    29.3 2038.11    78.6 2033.96   147.6 2031.97   203.4 2028.35
   236.1 2023.04   315.2 2000.86   331.8 1994.46   345.2 1992.92   355.3 1988.03
   419.2 1964.05     436 1954.56  447.531950.023   456.2 1946.87   496.3 1948.85
  510.271951.051     520  1953.3   691.5 1953.28     892  1950.7   916.7 1953.97
   923.4  1956.6   933.2 1968.67   946.9 1982.99   973.9  2005.7   987.3 2022.63
  1014.2 2038.63  1027.6 2049.93  1044.5 2058.06  1051.2 2063.85  1067.4  2068.5
#Mann= 4 ,-1 , 0
       0      .1       0  447.53    .045       0  510.27     .05       0
  798.67      .1       0
Bank Sta=447.53,510.27
XS Rating Curve= 0 ,0
Exp/Cntr=0.3,0.1

Type RM Length L Ch R = 1 ,52279   ,804.9,779,745.4
XS GIS Cut Line= 3
2150812.26291896371512.4312503042150312.26293471371450.972711816
2149999.76290356371443.681059733
#Sta/Elev= 30
       0 1981.57    76.1 1971.64   112.4 1963.16   132.3 1961.86   148.8 1953.08
   155.4 1952.03   337.2 1950.05     401 1951.61   408.9 1947.49   419.8 1943.61
  454.691946.527   505.8 1947.88     532 1946.78   541.9 1949.86   564.8 1944.68
   577.8 1947.62   584.5 1951.54   600.9 1952.59   607.5 1957.87   610.8 1962.96
   617.3  1977.2   620.6    1982   643.6 1999.96     660  2032.5   679.7 2044.04
   696.4 2050.01   725.3 2056.14   742.8  2064.1   761.7 2067.81   816.3 2072.67
#Mann= 5 ,-1 , 0
       0      .1       0  152.48     .05       0  308.32      .1       0
   408.9    .045       0  454.69      .1       0
Bank Sta=408.9,454.69
XS Rating Curve= 0 ,0
Exp/Cntr=0.3,0.1

Type RM Length L Ch R = 1 ,51500   ,617.6,594.2,572.5
XS GIS Cut Line= 3
2150520.59617947370436.3894391512150049.76280355371060.347836897
2149943.51268797371345.764588892
#Sta/Elev= 30
       0 2177.29    23.7 2154.22    48.9 2133.41    65.3 2121.99      77 2107.48
    89.5 2095.31   120.4 2072.08   216.9 2004.86   262.1 1975.57   297.2 1949.83
  330.331942.813   339.4 1940.52   364.9 1939.68  385.931942.459     398 1943.13
   410.1 1946.95   441.8 1949.42   615.6    1949   738.9 1951.47   779.5 1954.38
   790.8 1959.51   804.8 1960.54   825.5 1971.23   895.8 1998.09   916.8 2001.22
   927.3 2006.91   951.8 2014.05   997.3 2030.85  1028.8 2036.85  1086.2 2051.99
#Mann= 5 ,-1 , 0
       0      .1       0  330.33    .045       0  385.93      .1       0
  406.95    .055       0  701.54      .1       0
Bank Sta=330.33,385.93
XS Rating Curve= 0 ,0
Exp/Cntr=0.3,0.1

Type RM Length L Ch R = 1 ,50906   ,593.7,594.6,595.6
XS GIS Cut Line= 2
2149696.63785364370510.3479526492149834.13790672 371362.43122223
#Sta/Elev= 30
       0 2145.11    37.3 2111.99    60.6 2096.46    72.1 2082.15    97.2 2062.32
   110.4 2044.47   133.7 2025.38   160.3 2006.05     181 1985.43   206.9 1965.68
   226.8 1947.08   232.5 1943.63  238.66 1941.93     260 1937.87   286.6 1938.38
  294.241941.904   303.2 1944.02   333.1 1944.12   346.4 1947.72   542.5 1948.62
   602.3 1952.79   608.9 1955.02   615.6 1959.45   628.9  1960.8   645.5  1971.1
   665.4 1980.76   765.1 2023.68   833.5 2046.73   847.8 2048.69   863.1 2053.47
#Mann= 5 ,-1 , 0
       0      .1       0  238.66    .045       0  294.24      .1       0
  337.01    .055       0  561.56      .1       0
Bank Sta=238.66,294.24
XS Rating Curve= 0 ,0
Exp/Cntr=0.3,0.1

Type RM Length L Ch R = 1 ,50311   ,731.9,731.3,727.8
XS GIS Cut Line= 2
2149114.34603922370611.3894172312149274.76271313371573.889460728
#Sta/Elev= 30
       0 2094.03    14.8 2088.17      68 2072.05    91.3 2060.55   101.2 2052.63
   114.5 2045.71   131.2 2038.85   141.1 2029.15   161.1 2013.12   174.4 2006.85
   202.3 1986.85   217.6 1973.97   233.6 1963.12   247.6 1955.13   281.61940.875
   290.8 1938.24   314.1 1936.92   340.7 1937.65  356.911940.034     364  1940.2
   370.6 1942.88   377.3 1943.94   523.6 1943.55   783.1 1946.15     813 1949.92
   852.9  1960.9   879.5 1963.58   919.5 1963.77   949.4 1962.17   975.8 1962.68
#Mann= 6 ,-1 , 0
       0      .1       0   281.6    .045       0  356.91    .055       0
  424.34      .1       0  521.86     .05       0  656.34      .1       0
Bank Sta=281.6,356.91
XS Rating Curve= 0 ,0
Exp/Cntr=0.3,0.1

Type RM Length L Ch R = 1 ,49580   ,646.5,656.8,668.2
XS GIS Cut Line= 2
2148397.67949356370700.9728994822148626.84602997371660.347949222
#Sta/Elev= 30
       0 2046.57    27.4 2040.06      51 2031.76    73.8 2026.26    98.3 2014.54
   107.1 2004.79   117.3 1995.97   142.1 1980.42   162.4 1964.81   172.5 1953.25
  193.341939.283   199.5 1936.27   219.7 1935.21   250.1 1935.91  262.161939.426
   273.7 1941.28   337.9 1939.91   496.3 1943.47   745.9 1942.41   786.4 1944.86
     810 1952.43     828 1961.15   843.7 1976.28     864 1989.88   894.3 2006.93
   907.8  2019.5     927 2031.39     955 2045.42   965.2 2054.54   986.4 2063.94
#Mann= 6 ,-1 , 0
       0      .1       0  154.07      .1       0  193.34    .045       0
  262.16      .1       0  349.73     .05       0  741.03      .1       0
Bank Sta=193.34,262.16
XS Rating Curve= 0 ,0
Exp/Cntr=0.3,0.1

Type RM Length L Ch R = 1 ,48923   ,778.2,800.3,817.6
XS GIS Cut Line= 2
2147851.84626764370658.2646515672147751.84613955371533.264541984
#Sta/Elev= 30
       0 2024.09    69.8 2012.71   109.5 2007.83   149.1 1997.05   188.7 1979.86
   212.9  1965.9   238.3 1949.85   241.6 1946.75  248.821937.561   251.5 1934.31
   254.8 1932.72     268 1931.23   291.1 1931.95  307.751937.201   324.1 1937.78
   337.3  1940.5   350.5 1940.83   456.2 1938.94   633.7 1939.84   670.8 1942.15
     687 1944.62   710.7  1954.7   740.4 1972.21   766.1 1991.79   773.5  1999.2
   783.1 2005.83   789.7 2012.24   805.6 2020.93     850 2052.97   880.7 2071.89
#Mann= 5 ,-1 , 0
       0      .1       0   58.04      .1       0  248.82    .045       0
  307.75     .12       0  522.55      .1       0
Bank Sta=248.82,307.75
XS Rating Curve= 0 ,0
Exp/Cntr=0.3,0.1

Type RM Length L Ch R = 1 ,48123   ,417.2,411.1,406.1
XS GIS Cut Line= 2
2147511.22096464370478.0563505592146664.34601797371055.139513984
#Sta/Elev= 30
       0  2011.7    54.1 2004.25    94.3 2003.06   122.5 2000.15   162.8 1989.94
   195.8 1972.01   207.6 1962.82   225.7 1952.66   241.6 1938.74   249.5 1936.48
   524.8    1937  550.05 1931.24   577.2 1928.07  599.17 1933.72   604.3 1935.73
     618 1946.79   629.7 1949.18   646.5 1965.52   662.4 1976.29   690.2 1999.16
   717.1 2016.66   734.6 2034.02   771.9    2063     787 2072.35   805.3  2086.5
   829.2 2099.67   845.2 2112.87   908.6  2142.5   968.1 2172.39  1024.8 2188.07
#Mann= 6 ,-1 , 0
       0      .1       0   52.97      .1       0  237.92     .05       0
  446.18      .1       0  550.05    .045       0  599.17      .1       0
Bank Sta=550.05,599.17
XS Rating Curve= 0 ,0
Exp/Cntr=0.3,0.1

Type RM Length L Ch R = 1 ,47712   ,495.6,505.3,514.7
XS GIS Cut Line= 3
2147436.09086555370211.042448893 2146842.3410688370407.222830817
2146345.81319048370959.306044221
#Sta/Elev= 30
       0 2010.23    65.5 2001.61   106.9 1991.79   200.2  1959.9   283.2 1939.26
   349.9 1936.12   763.9 1934.08   787.1 1935.78  795.411933.134   803.4 1928.24
   813.6 1926.74   835.7 1927.36  847.751932.158   865.6 1936.41   875.4 1943.34
   889.3 1943.91     900 1948.88   923.9 1970.04     946 1981.44     959 1991.99
   984.6  2007.5  1012.8 2021.69  1075.2 2045.99  1144.5 2076.12  1179.8 2087.11
    1246 2102.05  1277.7 2106.15  1305.2 2106.71  1344.7 2111.72  1367.8 2112.44
#Mann= 5 ,-1 , 0
       0      .1       0  251.15     .05       0   763.9      .1       0
  795.41    .045       0  847.75      .1       0
Bank Sta=795.41,847.75
XS Rating Curve= 0 ,0
Exp/Cntr=0.5,0.3

Type RM Length L Ch R = 1 ,47206   ,59.6,63,72.6
XS GIS Cut Line= 6
2147342.47097406370180.1396235672146889.34622414370148.889686063
2146551.84624296370156.1813381462146353.53528789370216.394800395
2146261.63717772370417.9714969842146123.83331947370844.404043064
#Sta/Elev= 30
       0 1987.45    41.6 1973.41    57.3  1970.3     100 1965.64   182.2 1961.06
   221.7 1967.82   238.2  1967.4   248.3  1965.6   257.9 1962.11   264.5 1957.45
   297.8 1945.11   382.5 1937.51   484.7 1936.39   501.1  1936.1   691.5 1935.88
   792.8 1932.22   887.3 1932.72   938.7 1932.38  943.031931.605   956.8 1926.04
   977.5  1925.3 1006.721931.125  1046.5 1935.36  1126.7 1935.48  1189.9 1939.85
    1361 1940.88  1415.5 1943.05  1464.4 1943.69  1519.8 1951.47  1669.9 1993.05
#Mann= 9 ,-1 , 0
       0      .1       0   221.7     .06       0   484.7     .05       0
   501.1     .06       0   887.3     .05       0   938.7      .1       0
  943.03    .045       0 1006.72     .06       0  1415.5      .1       0
#XS Ineff= 3 ,-1
       0  923.03  1934.7 1026.72  1047.2  1934.7  1047.2 1669.88 1943.02
Permanent Ineff=
       F       F       F
Bank Sta=943.03,1006.72
XS Rating Curve= 0 ,0
Exp/Cntr=0.5,0.3

Type RM Length L Ch R = 1 ,47143   ,480.9,487.7,489
XS GIS Cut Line= 6
2147361.22126463370138.4727121442146875.80458455370109.306103811
2146539.34626797370100.9727871422146456.01277322370114.514426723
2146292.47110556370164.5146548152145800.80443797370429.097787067
#Sta/Elev= 30
       0 1987.24   113.3 1970.68   197.6 1983.72   210.8 1983.32   246.9  1988.9
   269.9 1987.64   292.7 1978.23   332.4 1967.41   381.7 1944.11   411.6 1937.67
   445.1 1938.91   552.5 1934.92   621.3 1936.81     733 1935.37   827.6 1930.24
  978.341931.639  1007.6  1924.4  1035.1 1927.15  1046.11931.722  1052.2 1935.04
  1121.2  1936.9  1132.5 1940.24  1143.8 1953.39  1176.1 1965.17  1230.1 1975.85
  1376.4 1994.83  1584.8 1995.22  1620.9 1993.46  1628.4 1989.62  1637.1 1988.88
#Mann= 6 ,-1 , 0
       0      .1       0  119.64     .06       0  978.34    .045       0
  1046.1     .06       0 1382.88      .1       0 1472.67     .06       0
Bank Sta=978.34,1046.1
XS Rating Curve= 0 ,0
Exp/Cntr=0.5,0.3

Type RM Length L Ch R = 1 ,46656   ,633.5,630.2,623.5
XS GIS Cut Line= 3
2146929.14634138369596.4590323872146019.42440756369716.250787556
 2145611.4380188369794.375631318
#Sta/Elev= 30
       0 2103.79     114 2059.04   152.7 2039.87   233.1 2006.46   284.3 1978.07
   299.3 1967.04   309.2 1953.22   345.6 1933.86   365.4 1936.23   378.7 1933.71
   448.2 1931.12   559.2  1931.5   626.9 1928.35   712.9 1930.58  720.951928.719
   729.5 1925.35   752.1 1922.84   762.5 1923.72  776.661928.235   798.9 1932.69
   894.9 1935.14   904.8 1942.05   941.5 1960.83   968.2 1978.27   981.5 1982.17
   998.3 1997.62  1044.9 2019.88  1098.2 2040.44  1227.2 2085.12    1333 2129.69
#Mann= 7 ,-1 , 0
       0      .1       0  346.81     .05       0  633.12      .1       0
  720.95    .045       0  776.66      .1       0  788.43     .06       0
  935.03      .1       0
Bank Sta=720.95,776.66
XS Rating Curve= 0 ,0
Exp/Cntr=0.3,0.1

Type RM Length L Ch R = 1 ,46025   ,399.6,393.4,393.1
XS GIS Cut Line= 2
2146821.50744906368945.4173554782145364.91029663369266.597815484
#Sta/Elev= 30
       0 2160.75      29  2144.2    99.5 2111.92   200.5 2077.55   261.1 2062.93
   351.9 2031.87   455.7  2011.3   485.9 1993.37     496 1982.35   514.3 1953.69
   539.6 1936.01   563.2 1932.22  580.241926.395     590 1921.73   600.1 1921.12
   640.4 1922.51  652.371926.547   660.2 1928.74   724.4 1925.62   919.3 1929.26
  1023.6 1928.75  1056.6 1930.28  1070.5  1934.6  1089.7 1935.19  1107.4 1948.76
  1120.9 1952.69  1174.6 1990.12  1235.5 2018.02  1335.9 2057.18  1491.6 2106.04
#Mann= 6 ,-1 , 0
       0      .1       0  509.09      .1       0  580.24    .045       0
  652.37     .05       0 1014.27     .06       0 1088.93      .1       0
Bank Sta=580.24,652.37
XS Rating Curve= 0 ,0
Exp/Cntr=0.3,0.1

Type RM Length L Ch R = 1 ,45632   ,632.2,637.9,643
XS GIS Cut Line= 2
2146677.41029631368589.5145239832145307.61874455368877.708829477
#Sta/Elev= 30
       0 2166.38    42.6 2154.56    92.9 2136.36   159.9 2105.05   183.4 2096.19
   253.2 2074.67   371.2    2042   455.4 2013.55     497 2001.33   508.6 1992.96
   522.3 1986.34   548.9 1961.49     579 1943.57   589.1 1933.69   605.8 1930.62
   616.31924.258     626 1918.57   629.3 1918.43   646.1 1919.34  662.19 1925.55
   669.5 1926.82   715.8 1924.57   779.5 1928.74  1095.3 1931.59  1156.2    1939
  1189.4 1962.09  1266.3  2001.8    1320 2033.43  1350.1 2054.84  1399.8 2083.69
#Mann= 7 ,-1 , 0
       0      .1       0  521.21      .1       0  575.09     .05       0
   616.3    .045       0  662.19     .05       0 1069.14     .06       0
 1196.92      .1       0
#XS Ineff= 1 ,-1
 1002.26 1399.78 1945.98
Permanent Ineff=
       F
Bank Sta=616.3,662.19
XS Rating Curve= 0 ,0
Exp/Cntr=0.3,0.1

Type RM Length L Ch R = 1 ,44994   ,688.7,699.1,702.2
XS GIS Cut Line= 2
2146593.15915248368108.3176517342145255.53551538368082.569999814
#Sta/Elev= 30
       0  2180.6      69 2144.75   269.2 2061.97   397.1 2005.43   469.8 1978.57
   491.5 1965.41   521.8 1940.09   533.3 1934.21   554.6  1927.6   607.2 1928.13
  623.031922.559   649.8 1916.65   659.7 1917.13  671.871922.473   692.5 1921.42
   727.4 1926.47   967.9 1925.68   994.4 1932.25  1010.8 1932.95  1023.9 1946.75
  1043.6 1958.62    1060 1976.86  1086.2 1997.25  1125.7 2021.58  1191.2 2075.61
  1243.8 2102.79  1263.4 2122.01  1302.8 2152.55  1319.2 2162.79  1337.9  2169.2
#Mann= 6 ,-1 , 0
       0      .1       0  523.01      .1       0  623.03    .045       0
  671.87     .05       0  957.88     .06       0 1095.12      .1       0
Bank Sta=623.03,671.87
XS Rating Curve= 0 ,0
Exp/Cntr=0.3,0.1
